--- PnyCrk.prj (project) ---

Proj Title=PnyCrk
Current Plan=p01
Default Exp/Contr=0,0
English Units
Geom File=g01
Flow File=f01
Plan File=p01
BEGIN DESCRIPTION:
END DESCRIPTION:
DSS Export Rating Curves= 0
DSS Export Rating Curve Sorted= 0
DSS Export Volume Flow Curves= 0
DXF OffsetX= 0
DXF OffsetY= 0
DXF ScaleX= 0
DXF ScaleY= 0

--- PnyCrk.p01 (plan) ---

Plan Title=Floodplain
Program Version=4.00
Geom File=g01
Flow File=f01
K Sum by GR=0
Std Step Tol=0.01
Critical Tol=0.01
Num of Std Step Trials=20
Max Error Tol=0.3
Flow Tol Ratio=0.001
Split Flow NTrial=30
Split Flow Tol=0.02
Split Flow Ratio=0.02
Log Output Level=0
Friction Slope Method=1
Unsteady Friction Slope Method=2
Unsteady Bridges Friction Slope Method=1
Global Log Level=0
CheckData=False
Run HTab=0
Run UNet=0
Run PostProcess=0
UNET Theta=0
UNET Theta Warmup=0
UNET ZTol=0
UNET ZSATol=0
UNET MxIter=0
UNET MaxInSteps=0
UNET DtIC=0
UNET DtMin=0
UNET MaxCRTS=0
UNET WFStab=0
UNET SFStab=0
UNET WFX=0
UNET SFX=0
UNET DSS MLevel=0
UNET DZMax Abort=0
UNET Convert EG Bridges=0
UNET Use Existing IB Tables=0
UNET Froude Limit=0
UNET Froude Power=0
Write IC File=0
Echo Input=False
Echo Output=False
Write Detailed=0

--- PnyCrk.f01 (steady flow) ---

Flow Title=NFF Regression Equation
Program Version=4.00
Number of Profiles=1
Profile Names=P100yr
River Rch & RM=PnyCrk,Main      ,63478.1
11080.04
River Rch & RM=PnyCrk,Main      ,57127.2
11157.84
River Rch & RM=PnyCrk,Main      ,56691.8
11157.84
River Rch & RM=PnyCrk,Main      ,34298.9
11499.16
River Rch & RM=PnyCrk,Main      ,33861.5
12844.04
River Rch & RM=PnyCrk,Main      ,13525.7
13548.08
River Rch & RM=PnyCrk,Main      ,11878.1
14454.87
River Rch & RM=PnyCrk,Main      ,620.7
15122.14
Boundary for River Rch & Prof#=PnyCrk,Main      ,1
Up Type=0
Dn Type=3
Dn Slope=0.01068

--- PnyCrk.g01 (geometry) ---

Geom Title=USGS 3m DEM
Program Version=4.10

River Reach=PnyCrk          ,Main
Reach XY= 30
     1923218.046      275863.938      1923989.35      276776.538
     1925061.093      276931.694     1923690.508      278336.355
     1924573.093      280478.602     1923377.726      280934.294
     1923441.341      281722.959     1924217.536      282011.542
     1924949.677       281514.53     1926024.777      282685.896
     1927889.018      282598.867     1928201.675      280978.552
      1929025.02      281750.446      1928468.28      283578.377
      1929012.87       289074.86      1928613.83       290003.11
     1926323.384       291498.75     1929990.348      292532.963
     1928117.991      296069.604     1929002.812      298996.257
     1930497.685      300469.914     1933333.027      300251.385
     1935044.945       301053.93     1937321.381       300531.39
     1939086.585      301141.989     1939353.792       303111.06
     1940545.188      305582.576       1941735.7      305551.306
     1940861.736      307240.086     1941938.631      309627.305

Type RM Length L Ch R = 1 ,63478.1 ,404,399.9,395.7
XS GIS Cut Line= 3
     1923090.615      276462.191     1923407.073      276202.481
     1923725.312      275944.127
#Sta/Elev= 30
       0 2156.97    69.9 2155.74    79.9 2153.07    89.9 2146.85    99.8 2137.32
   129.8  2120.9   139.8 2118.92   169.7 2118.71   179.7  2116.8   189.7 2112.45
   199.7 2102.24   209.7 2094.73   219.7 2089.89   229.6 2087.44   329.5 2081.67
   369.4  2070.7   396.9 2070.38   419.4 2070.28   421.9  2070.3   439.4 2070.84
   479.4 2077.53   529.4 2082.36   559.4 2094.56   599.3 2098.57   619.3 2107.02
   689.3 2129.82   729.3 2146.78   759.3 2163.53   809.3  2201.9   819.3 2213.05
#Mann= 3 , 0 , 0
       0      .1       0   396.9    .045       0   421.9      .1       0
Bank Sta=396.9,421.9
XS Rating Curve= 0 ,0
Exp/Cntr=0.3,0.1

Type RM Length L Ch R = 1 ,63078.1 ,493.4,475.3,457.3
XS GIS Cut Line= 3
     1923412.545      276790.528     1923687.536      276487.098
     1923962.528      276183.668
#Sta/Elev= 30
       0 2211.94      40 2195.97    59.9 2191.62    99.9 2171.96   109.9 2163.45
   149.8 2122.99   159.8 2114.82   169.8 2110.69   179.8  2109.2   189.8 2103.34
   209.7 2088.15   219.7  2083.2   349.6 2079.26   379.5 2067.91     397 2066.62
   399.5  2066.6     422 2066.66   439.5  2067.5   449.4  2071.1   469.4 2083.57
   489.4 2090.44   509.4 2092.11   559.3 2102.13   659.2 2128.09   679.2 2130.45
   699.2 2135.85   729.1 2147.56     789 2178.43     799  2179.5     819 2189.87
#Mann= 3 , 0 , 0
       0      .1       0     397    .045       0     422      .1       0
Bank Sta=397,422
XS Rating Curve= 0 ,0
Exp/Cntr=0.3,0.1

Type RM Length L Ch R = 1 ,62602.4 ,285.8,279.7,273.5
XS GIS Cut Line= 3
     1923974.864      277051.315     1924030.981      276872.441
     1924083.591      276314.774
#Sta/Elev= 30
       0 2237.63    29.6  2231.4    39.5  2226.9    69.1 2211.58   108.5 2184.71
   118.4 2184.31   128.3 2177.78     148 2161.12   157.9 2149.87   177.6 2120.23
   187.5 2111.37   217.5 2098.86   237.5  2076.1   247.5    2068   257.5 2063.44
   262.6 2062.86   267.5 2062.31   287.6 2063.33   307.5 2065.38   347.5 2073.57
   437.5 2074.06   447.5  2075.3   477.5 2084.77   517.6 2087.52   587.6 2096.48
   607.6 2101.72   657.6 2121.14   667.6 2124.27   677.6 2125.12   747.6 2153.38
#Mann= 3 , 0 , 0
       0      .1       0   262.6    .045       0   287.6      .1       0
Bank Sta=262.6,287.6
XS Rating Curve= 0 ,0
Exp/Cntr=0.3,0.1

Type RM Length L Ch R = 1 ,62322.5 ,432.3,434,435.7
XS GIS Cut Line= 3
     1923918.495       277168.67      1924336.12      276904.007
     1924266.992      276372.927
#Sta/Elev= 30
       0 2278.12    39.6 2270.77    79.1 2260.31   158.2 2260.79     178  2263.4
   247.2 2253.33     267 2255.47   276.9 2252.82   405.4 2197.44   415.3 2194.37
   435.1 2194.83   494.4 2174.83   504.3 2162.56   534.1 2119.58     544  2113.6
   553.9 2112.41   563.8  2106.2   603.5 2070.58   613.4 2065.43   633.3 2062.07
   637.9 2062.07   662.9  2062.1   702.7 2067.46     782 2071.95   821.7 2081.18
   851.5 2083.36     911 2103.14   930.8 2107.35  1000.2 2137.51    1030 2145.65
#Mann= 3 , 0 , 0
       0      .1       0   637.9    .045       0   662.9      .1       0
Bank Sta=637.9,662.9
XS Rating Curve= 0 ,0
Exp/Cntr=0.3,0.1

Type RM Length L Ch R = 1 ,61888.6 ,374.6,410.4,449.1
XS GIS Cut Line= 3
     1923986.645      277167.989     1924749.986      276837.368
     1924716.074      276331.805
#Sta/Elev= 30
       0 2255.26    19.8  2251.7      99 2252.58   188.2 2267.77   247.6 2265.17
   336.7 2243.39   356.5 2234.44   445.6 2205.27   534.8 2181.55   673.4 2151.51
   703.1  2141.2   812.1 2115.39   831.9 2111.97   861.7 2111.19   901.4 2098.58
   911.4 2098.18   931.2 2087.35     961 2066.59     971 2063.03   990.8  2062.1
  1006.7  2062.1  1031.7  2062.1  1100.1 2067.26  1149.8 2079.43  1169.7 2094.05
  1189.5 2102.02    1269 2163.78  1288.9 2170.38  1308.8 2182.82  1338.6 2196.55
#Mann= 3 , 0 , 0
       0      .1       0  1006.7    .045       0  1031.7      .1       0
Bank Sta=1006.7,1031.7
XS Rating Curve= 0 ,0
Exp/Cntr=0.3,0.1

Type RM Length L Ch R = 1 ,61478.1 ,368.6,399,426.5
XS GIS Cut Line= 3
     1924041.425      277215.886     1925047.999      276842.749
     1925331.211      276770.338
#Sta/Elev= 30
       0 2229.55    29.8  2228.3    79.5 2231.52   188.9 2249.89   228.6 2247.33
   268.4 2239.71   437.4 2198.72   636.2 2140.16   745.5 2116.99   795.2 2103.64
     835 2103.07   864.8  2092.9   884.6 2081.37   894.6 2078.52     994 2074.47
  1053.6 2060.12    1061 2060.15    1086 2060.33  1102.7 2063.58    1132 2075.18
  1141.7  2084.5  1190.4 2141.76  1209.9 2166.64  1219.7 2185.34  1229.4 2193.17
  1248.9 2206.26  1297.6 2232.68  1317.1 2250.15  1336.6 2263.08  1365.8  2276.2
#Mann= 3 , 0 , 0
       0      .1       0    1061    .045       0    1086      .1       0
Bank Sta=1061,1086
XS Rating Curve= 0 ,0
Exp/Cntr=0.3,0.1

Type RM Length L Ch R = 1 ,61078.4 ,397.5,401,404.5
XS GIS Cut Line= 3
     1924030.612      277291.384     1924746.479      277019.749
     1925177.918      277417.314
#Sta/Elev= 30
       0  2231.6    29.8  2222.1    39.8 2216.08    69.6  2208.5    99.4 2210.12
     179 2223.78   248.6 2226.71   278.4 2225.33   367.9 2210.88   467.4 2185.66
     537 2173.16   795.5 2099.51   835.3 2092.35     875 2075.89   924.8 2072.34
   984.4 2057.28  1004.3 2055.44  1019.8 2055.46  1044.8 2055.89  1073.9 2067.06
  1093.8 2069.95  1103.8 2077.99  1123.6 2112.73  1153.5 2137.72  1163.4 2148.96
  1223.1 2193.35    1243 2205.28  1262.9 2222.58  1272.8 2234.67  1352.4 2292.84
#Mann= 3 , 0 , 0
       0      .1       0  1019.8    .045       0  1044.8      .1       0
Bank Sta=1019.8,1044.8
XS Rating Curve= 0 ,0
Exp/Cntr=0.3,0.1

Type RM Length L Ch R = 1 ,60677.4 ,409.3,420.1,430.8
XS GIS Cut Line= 3
     1923985.785      277355.967     1924465.892      277254.741
     1924882.153      277750.654
#Sta/Elev= 30
       0 2247.28    68.7 2223.15    88.3 2213.35   166.8 2191.74   225.7 2191.29
     265 2195.73   294.4 2195.14   402.3 2176.18   480.8 2157.69   490.7 2152.76
   570.4  2093.1   590.3 2085.34   610.2 2072.13   630.1 2068.81   709.8 2068.84
   719.8 2067.16   749.6 2052.14   759.6  2050.5   762.7  2050.5   787.7 2050.55
   819.4 2057.52   829.3 2062.53   849.2 2065.81   859.2 2070.36   938.9 2124.07
  1008.6 2163.92  1028.6 2165.16  1058.4 2160.85  1078.4 2163.24  1138.1 2185.18
#Mann= 3 , 0 , 0
       0      .1       0   762.7    .045       0   787.7      .1       0
Bank Sta=762.7,787.7
XS Rating Curve= 0 ,0
Exp/Cntr=0.3,0.1

Type RM Length L Ch R = 1 ,60257.4 ,392,379.2,366.5
XS GIS Cut Line= 3
     1923924.354      277421.232     1924220.378      277444.138
     1924428.339      278072.401
#Sta/Elev= 30
       0 2262.78    19.8 2253.49    49.5 2243.71    69.3 2234.57   128.7 2216.29
   148.4 2208.34   207.8 2190.93   247.4 2170.91     287 2155.02   296.9 2149.82
   346.3 2108.18   356.2 2102.13     366 2099.31   395.7 2076.27   415.4 2065.78
   435.2 2060.45   474.7 2056.65     537 2046.56   543.8  2046.5     562  2046.5
   583.4 2047.37   642.6 2057.05     692 2061.09   701.9 2063.48   741.4 2079.83
   761.2 2084.23     850 2116.07   879.7 2131.69   938.9 2167.95   958.7 2173.99
#Mann= 3 , 0 , 0
       0      .1       0     537    .045       0     562      .1       0
Bank Sta=537,562
XS Rating Curve= 0 ,0
Exp/Cntr=0.3,0.1

Type RM Length L Ch R = 1 ,59878.1 ,405.5,400,394
XS GIS Cut Line= 3
     1923713.118      277612.393     1924001.333      277903.292
     1924289.873       278193.87
#Sta/Elev= 30
       0 2295.99      20 2292.66      30 2287.81    89.9 2244.28   109.9 2235.22
   149.8 2204.36   169.8 2183.86   209.7 2151.63   219.7 2143.94   229.7 2140.25
   239.7 2133.48   269.7 2109.22   289.6 2088.52   319.6 2064.71   359.6 2047.73
     397 2042.45   399.5 2042.44     422 2043.24   449.4 2047.64   489.4 2058.99
   519.4 2063.92   579.3 2055.84   619.2 2056.92   669.2 2066.35   689.2 2075.07
   709.1 2087.27   729.1 2100.17   749.1 2118.78   769.1 2128.15     819 2161.74
#Mann= 3 , 0 , 0
       0      .1       0     397    .045       0     422      .1       0
Bank Sta=397,422
XS Rating Curve= 0 ,0
Exp/Cntr=0.3,0.1

Type RM Length L Ch R = 1 ,59478.1 ,415.1,400,385.5
XS GIS Cut Line= 3
     1923417.334      277991.741     1923757.553      278219.616
     1924102.286      278440.814
#Sta/Elev= 30
       0 2284.55      40 2279.64    59.9 2273.16    99.9 2247.03   109.9 2235.09
   199.8    2166   219.7 2142.26   259.7 2110.45   279.6 2098.24   299.6 2083.15
   309.6 2071.46   319.6 2062.48   329.6    2057   369.5 2042.87     397 2039.37
   399.5 2039.35     422 2041.02   449.4 2048.17   489.4 2061.85   519.4  2075.1
   539.4 2078.86   579.3 2068.87   609.3 2058.95   649.2 2052.89   679.2 2052.27
   689.2 2053.74   759.1 2067.24   789.1 2080.37   799.1 2088.71   819.1 2100.47
#Mann= 3 , 0 , 0
       0      .1       0     397    .045       0     422      .1       0
Bank Sta=397,422
XS Rating Curve= 0 ,0
Exp/Cntr=0.3,0.1

Type RM Length L Ch R = 1 ,59078.1 ,416.7,413,409.4
XS GIS Cut Line= 3
     1923252.481      278580.658     1923661.568      278599.037
     1924070.655      278617.417
#Sta/Elev= 30
       0  2315.6    49.9 2310.87    59.9 2307.23    89.9 2289.58   109.9 2270.32
   169.8 2227.03   189.8 2202.74   249.7  2148.7   269.7 2120.56   309.6 2085.08
   349.6 2052.59     397 2037.69   419.5 2035.23     422 2035.23   439.5 2035.83
   449.4 2038.14   499.4 2055.51   519.4 2065.46   559.3  2078.1   569.3 2078.85
   579.3  2076.4   599.3 2064.06   609.3 2061.31   639.2  2057.2   659.2 2051.14
   669.2 2049.65   689.2 2051.53   749.1 2062.69     789 2079.25     819 2094.34
#Mann= 3 , 0 , 0
       0      .1       0     397    .045       0     422      .1       0
Bank Sta=397,422
XS Rating Curve= 0 ,0
Exp/Cntr=0.3,0.1

Type RM Length L Ch R = 1 ,58665.1 ,646.6,633.1,619.7
XS GIS Cut Line= 3
     1923281.627      279046.528     1923789.759      279001.871
     1924090.305      278910.114
#Sta/Elev= 30
       0 2303.54      10 2294.42      70 2258.99      90 2237.86     150 2199.96
     160 2191.65     170 2181.14     230 2148.91     250 2133.35     310 2103.61
   320.1 2092.41   330.1 2072.49   340.1 2061.65   350.1 2053.48   380.1 2039.55
   396.8 2034.53   420.1 2033.69   421.8 2033.71   440.1 2034.83   490.1 2052.44
   549.4 2064.69   559.2 2064.69   578.8  2057.4   608.3  2051.1   637.8 2048.02
   657.4 2047.98   726.1 2068.15   775.2 2099.04   794.9  2108.5   824.3 2111.37
#Mann= 3 , 0 , 0
       0      .1       0   396.8    .045       0   421.8      .1       0
Bank Sta=396.8,421.8
XS Rating Curve= 0 ,0
Exp/Cntr=0.3,0.1

Type RM Length L Ch R = 1 ,58031.8 ,150.8,153.6,157.8
XS GIS Cut Line= 3
      1923634.87      279712.196     1924194.327      279342.076
     1924428.793      279135.195
#Sta/Elev= 30
       0 2158.09    49.3 2142.84    59.2 2138.15    78.9 2114.85   108.5 2089.27
   128.2 2069.61   138.1 2062.04   157.8 2055.53   177.6  2045.7   197.3 2039.25
   226.9 2030.47   246.6  2028.6   266.4 2028.81   315.7 2035.25   384.7 2034.18
   443.9  2029.7   478.3 2029.21   503.3 2029.74     513 2032.63   532.7 2044.57
   562.3 2055.32   572.2 2064.77     582 2077.67   591.9 2084.74   719.7 2101.25
     749 2101.46   778.3 2107.56   846.7 2110.74   944.4 2119.02   983.5 2127.89
#Mann= 3 , 0 , 0
       0      .1       0   478.3    .045       0   503.3      .1       0
Bank Sta=478.3,503.3
XS Rating Curve= 0 ,0
Exp/Cntr=0.3,0.1

Type RM Length L Ch R = 1 ,57878.1 ,401.7,399.5,398.4
XS GIS Cut Line= 3
     1923709.696      279791.196     1924111.484      279579.465
     1924476.535      279412.027
#Sta/Elev= 30
       0 2128.95    19.8  2121.8    29.6 2115.07    59.2 2093.35    69.1 2084.17
      79 2072.11   108.6 2051.64   128.4 2043.84     158 2034.75   167.8 2028.81
   187.6 2026.08   227.1  2026.3     237 2027.32   256.7 2034.74   325.8 2035.27
   355.4 2033.51   414.7 2026.02   441.7 2026.65   466.7 2027.72   473.8 2028.94
   503.1 2044.02   542.3 2054.59   552.1 2058.82   571.7 2071.92   620.7 2089.85
   659.9 2097.83   767.6 2112.43   806.8  2120.4   836.2 2121.11   855.8 2126.18
#Mann= 3 , 0 , 0
       0      .1       0   441.7    .045       0   466.7      .1       0
Bank Sta=441.7,466.7
XS Rating Curve= 0 ,0
Exp/Cntr=0.3,0.1

Type RM Length L Ch R = 1 ,57478.1 ,354,350.8,345
XS GIS Cut Line= 3
     1923840.528      280175.831     1924183.116      279959.562
     1924569.401      279760.994
#Sta/Elev= 30
       0 2090.46    39.5 2086.26   158.1 2078.98     168 2080.02   197.6 2088.51
   217.4 2089.47     247 2089.03   256.9 2086.69   266.8 2080.43   296.4  2054.9
   306.3 2048.67   316.2  2044.1   326.1 2042.62     336 2039.66   365.6 2027.44
   375.5 2024.22   392.6 2022.62   395.3  2022.6   417.6  2022.6   454.5 2023.48
   503.8 2032.32   582.8 2043.32   602.6 2050.17   612.4 2054.57   671.7 2084.01
   681.5 2091.52   760.5 2121.95   770.4 2129.19   780.2 2133.15   839.5 2153.52
#Mann= 3 , 0 , 0
       0      .1       0   392.6    .045       0   417.6      .1       0
Bank Sta=392.6,417.6
XS Rating Curve= 0 ,0
Exp/Cntr=0.3,0.1

Type RM Length L Ch R = 1 ,57127.2 ,402.7,434.6,466.6
XS GIS Cut Line= 3
     1923892.786      280265.115     1924287.424      280323.039
     1924727.763      279967.499
#Sta/Elev= 30
       0 2089.53    29.9 2081.49    59.8 2079.92   259.3 2076.94   329.1 2079.71
     339 2077.81     349  2073.6   378.9 2057.78   388.9 2050.39   468.4 2042.99
     518 2035.28   527.9 2032.21   547.8 2022.03   567.7 2020.34   568.8 2020.35
   593.8 2020.63   617.3 2022.27     657  2036.7   696.7  2047.6   706.7 2051.48
   736.5 2070.52   756.3 2079.85   786.1 2099.21     796 2109.69   855.6 2156.62
   895.3 2190.97   905.2 2201.76   925.1 2218.95     945 2235.18   964.8 2248.56
#Mann= 3 , 0 , 0
       0      .1       0   568.8    .045       0   593.8      .1       0
Bank Sta=568.8,593.8
XS Rating Curve= 0 ,0
Exp/Cntr=0.3,0.1

Type RM Length L Ch R = 1 ,56691.8 ,502.5,516.5,530.5
XS GIS Cut Line= 3
     1923898.006      280352.145     1924287.424      280454.064
     1924866.585       280749.34
#Sta/Elev= 30
       0 2088.25    19.6 2080.41    39.3 2075.18     108 2071.38     216 2069.01
   255.3 2064.93   294.5  2063.4   382.9 2051.97   432.5 2043.46   482.5 2036.78
   532.6 2032.57   612.6 2028.37   652.6 2020.16   662.6 2019.39     679  2019.4
   692.6 2020.36     704 2024.54   722.6 2033.24   742.6 2037.77   752.6 2042.86
   802.6 2081.38   842.6 2115.82   852.6  2132.5   882.6 2168.82   922.6 2231.96
   942.6 2252.26   982.6 2276.69  1002.6 2283.28  1022.6 2283.92  1052.6 2277.26
#Mann= 3 , 0 , 0
       0      .1       0     679    .045       0     704      .1       0
Bank Sta=679,704
XS Rating Curve= 0 ,0
Exp/Cntr=0.3,0.1

Type RM Length L Ch R = 1 ,56174.9 ,664,666.8,669.6
XS GIS Cut Line= 3
      1923851.81      280442.032     1924204.671      280988.508
      1924294.32      281085.053
#Sta/Elev= 30
       0 2084.89    90.1 2077.68   110.1 2072.54   140.1 2061.31   150.1 2060.22
   190.2 2045.43   230.2 2037.61   320.2 2030.86   420.3 2026.04   430.3  2024.2
   450.3 2015.08   470.4  2012.7   471.5 2012.71   496.5  2013.1   510.4 2014.41
   540.4 2027.72   560.4 2042.28   590.4 2069.03   600.5 2072.61   610.5 2078.13
   640.5 2105.85   678.7 2143.57   697.6 2164.47     707 2176.24   716.4 2180.78
   725.8 2188.13   735.2 2198.33     754  2207.8   772.8 2220.48   782.2 2224.61
#Mann= 3 , 0 , 0
       0     .06       0   471.5    .045       0   496.5      .1       0
Bank Sta=471.5,496.5
XS Rating Curve= 0 ,0
Exp/Cntr=0.3,0.1

Type RM Length L Ch R = 1 ,55507.6 ,411.8,386.5,361.2
XS GIS Cut Line= 3
     1923330.359      280662.445     1923570.235      281109.189
     1923615.059      281140.221
#Sta/Elev= 30
       0 2201.54    19.9 2182.09    49.7 2150.88    79.5  2120.8    89.5 2111.69
    99.4 2110.36   109.4  2096.7   119.3 2076.09   129.2  2053.5   139.2  2032.4
   149.1 2017.94   159.1 2011.04     169 2008.57   198.8  2007.1   247.2  2007.1
   272.2 2007.81   278.4 2008.81   288.3  2012.2   298.3 2016.69   308.2 2019.68
   328.1 2021.95   387.8 2024.59   397.7 2026.47   407.6 2029.45   417.6 2030.43
   437.5 2035.69   457.4 2039.36   477.2 2044.89   525.2 2054.02   561.6 2061.87
#Mann= 3 , 0 , 0
       0     .06       0   247.2    .045       0   272.2      .1       0
Bank Sta=247.2,272.2
XS Rating Curve= 0 ,0
Exp/Cntr=0.3,0.1

Type RM Length L Ch R = 1 ,55120.8 ,461.3,442.7,423.5
XS GIS Cut Line= 2
     1923031.824      281167.323     1923580.579      281257.454
#Sta/Elev= 30
       0 2118.19     9.9 2110.53    29.8 2099.28    39.7 2091.02    49.6 2080.71
   109.2 2038.99   119.2 2031.42   129.1 2020.74     149 2010.86   158.9 2007.31
   178.8 2003.38   188.7 2002.41   208.5 2001.95   218.3 2002.02   238.3 2002.47
   243.3 2003.26   258.2 2006.62     278 2012.45     288 2016.12   347.6 2019.78
   357.5 2021.24   367.4 2024.08   377.4 2025.85   446.9 2030.44   456.8 2032.62
   466.7 2035.77   516.4 2053.98   526.3 2058.65   536.2 2064.28   556.1 2070.72
#Mann= 3 , 0 , 0
       0      .1       0   218.3    .045       0   243.3      .1       0
Bank Sta=218.3,243.3
XS Rating Curve= 0 ,0
Exp/Cntr=0.3,0.1

Type RM Length L Ch R = 1 ,54678.1 ,424.6,408.3,392.5
XS GIS Cut Line= 3
      1923168.76      281720.072       1923370.1      281609.621
     1923921.933      281291.934
#Sta/Elev= 30
       0 2162.66      10 2151.34      30 2124.53    39.9 2113.09    79.9 2076.68
    89.9  2062.3    99.8 2054.26   119.8 2043.53   179.7 2000.01   189.7 1997.44
   217.1  1996.2   242.1  1996.2   259.5 1996.16   269.4  1998.5   289.3 2007.28
   299.3 2009.19   329.1 2008.69   339.1  2010.4   368.9 2023.52   398.8 2027.02
   408.7 2029.76   438.6 2041.79   458.5 2053.32   468.4  2057.1   617.7 2076.51
   667.4 2087.26   717.2 2102.01   816.6 2136.48   826.6 2142.71   866.4 2155.41
#Mann= 3 , 0 , 0
       0      .1       0   217.1    .045       0   242.1      .1       0
Bank Sta=217.1,242.1
XS Rating Curve= 0 ,0
Exp/Cntr=0.3,0.1

Type RM Length L Ch R = 1 ,54269.8 ,360.3,349.6,338.9
XS GIS Cut Line= 2
      1923559.64       282088.27     1923832.285       281560.88
#Sta/Elev= 30
       0 2142.79    19.8 2126.83    39.6 2107.22    49.5 2104.34    59.4 2098.33
   108.8 2059.14   138.5 2033.09   158.3 2024.47     188 2001.56   197.9 1996.88
   207.8 1995.32   238.8 1992.83   263.8 1991.39   296.8  1991.1   306.7 1993.46
   326.5 2004.99   336.4 2007.96   346.3 2008.21   366.1 2012.87     376  2017.7
   395.8 2029.21   405.7 2033.97   415.6 2037.89   435.4 2044.26   455.2 2048.64
     475 2051.29   514.5 2059.24   544.2 2066.49   554.1 2068.22   593.7 2072.76
#Mann= 3 , 0 , 0
       0      .1       0   238.8    .045       0   263.8      .1       0
Bank Sta=238.8,263.8
XS Rating Curve= 0 ,0
Exp/Cntr=0.3,0.1

Type RM Length L Ch R = 1 ,53919.7 ,490.5,464.2,437.8
XS GIS Cut Line= 2
     1923977.477      282269.121     1924039.166      281581.568
#Sta/Elev= 30
       0 2173.72      20 2145.35      30 2135.37      40 2132.76      60 2111.24
      90 2092.63     120 2069.52   130.1 2067.48   160.1 2036.75   190.1 2012.42
   220.1  1994.7   230.1 1994.06   250.1 1988.34   271.3  1988.2   296.3 1988.19
   340.2 1987.81   350.2 1988.78   370.2 1995.06   390.2 1996.81   400.2 2001.38
   410.2 2001.71   420.2  2005.9   450.2 2008.73   490.2 2024.37   500.2 2024.36
   550.2 2037.37   600.3    2041   650.3 2059.46   680.3 2073.12   690.3 2073.23
#Mann= 3 , 0 , 0
       0      .1       0   271.3    .045       0   296.3      .1       0
Bank Sta=271.3,296.3
XS Rating Curve= 0 ,0
Exp/Cntr=0.3,0.1

Type RM Length L Ch R = 1 ,53455.3 ,259,263.8,268.6
XS GIS Cut Line= 2
     1924663.077      282089.616     1924094.334      281605.705
#Sta/Elev= 30
       0 2207.65    39.8  2200.7    59.7 2202.39    99.6 2196.92   109.5 2195.04
   119.5 2188.72   129.4 2177.37   139.4 2164.04   159.3 2135.06   169.3 2114.64
   179.2 2092.99   199.1  2071.9     219 2043.74     229 2030.93   248.9 2008.43
   258.9 1998.37   268.8 1989.76   278.8 1985.25   315.2 1984.61   328.6 1984.56
   340.2 1984.63   378.4 1984.93   418.2 1986.54   497.8 1997.18   567.5 2003.82
   587.4 2008.67   617.3 2018.91   627.3 2020.68     697 2042.83   746.8  2059.7
#Mann= 3 , 0 , 0
       0      .1       0   315.2    .045       0   340.2      .1       0
Bank Sta=315.2,340.2
XS Rating Curve= 0 ,0
Exp/Cntr=0.3,0.1

Type RM Length L Ch R = 1 ,53191.3 ,466.5,503.5,540.7
XS GIS Cut Line= 3
     1924859.796      282005.675     1924373.624      281422.959
     1924390.865      281216.078
#Sta/Elev= 30
       0 2132.87    39.9 2127.21    59.9 2127.36   149.8 2109.05   189.7 2105.77
   229.7 2095.23   279.6 2071.49   289.6 2071.63   299.6 2065.82   309.6 2054.34
   339.5 2011.12   349.5 1998.58   359.5 1988.85   369.5 1984.06   379.4 1981.76
   406.9 1979.51   429.4  1979.4   431.9  1979.4   489.3 1980.47   589.1 1998.11
   639.1 2000.71     669 2006.82   768.8 2055.22   778.7 2056.09   788.6 2059.83
   808.3 2070.53   857.8 2104.72   877.5 2112.05   946.7 2168.07   966.5 2175.08
#Mann= 3 , 0 , 0
       0      .1       0   406.9    .045       0   431.9      .1       0
Bank Sta=406.9,431.9
XS Rating Curve= 0 ,0
Exp/Cntr=0.3,0.1

Type RM Length L Ch R = 1 ,52687.3 ,429.4,424.3,419.2
XS GIS Cut Line= 3
     1924917.952      282049.415      1924904.62      281705.697
     1925253.972      281246.107
#Sta/Elev= 30
       0 2136.25    39.3  2122.9    78.6 2111.97    88.4 2111.91   167.1 2094.06
   176.9 2093.82   196.6 2089.31   206.4 2084.36   255.5 2050.38   265.4 2048.51
   275.2 2043.96     344 1997.23   353.9 1994.39   443.5 1980.34   473.4 1971.97
   503.2 1967.35   514.3 1967.41   539.3 1969.48     553 1975.71   572.9 1988.87
   612.7 1994.09   642.6 2001.77   702.3 2024.53   712.2 2025.42   722.2 2028.75
     772 2048.76   811.8 2069.61   831.7 2076.26   911.3  2121.3   921.3  2128.4
#Mann= 3 , 0 , 0
       0      .1       0   514.3    .045       0   539.3      .1       0
Bank Sta=514.3,539.3
XS Rating Curve= 0 ,0
Exp/Cntr=0.3,0.1

Type RM Length L Ch R = 1 ,52262.9 ,364.2,384.5,407.2
XS GIS Cut Line= 3
     1925050.386      282097.517     1925266.663      281864.306
     1925539.057      281312.623
#Sta/Elev= 30
       0 2109.67    49.7 2097.55    69.6  2088.1    89.4 2073.28   109.3 2063.47
   198.8 2029.56   308.1  2014.9   347.8 2007.06   377.6 1999.14   397.4 1989.97
     457 1982.57   486.8 1966.13   501.8  1964.6   506.6 1964.44   526.8 1964.84
   536.4 1967.93   546.3  1976.1   566.2 1997.24   576.1 2004.93   595.9 2019.12
   615.8 2026.93   695.2 2086.65     715 2094.47   794.4 2143.51   824.2 2157.63
     844 2171.36   893.6 2189.34   913.5  2199.2   923.4 2200.99   933.3 2207.36
#Mann= 3 , 0 , 0
       0      .1       0   501.8    .045       0   526.8      .1       0
Bank Sta=501.8,526.8
XS Rating Curve= 0 ,0
Exp/Cntr=0.3,0.1

Type RM Length L Ch R = 1 ,51878.1 ,392.9,406.5,417.8
XS GIS Cut Line= 3
     1925104.712      282186.657     1925496.242      282023.516
     1925884.171      281900.677
#Sta/Elev= 30
       0 2083.45    39.5 2070.67    98.6 2040.17   157.8  2028.3   187.4 2018.16
   256.5 2005.29   295.9 1987.68   335.4 1980.38   374.8 1964.61   384.7 1962.19
   411.7 1961.81   436.7 1961.81   473.8 1961.52   503.6 1965.04   553.2  1993.7
   563.1 2003.98   592.9 2049.16   602.8 2071.28   612.7 2088.27   622.6 2100.67
   642.5 2122.19   672.3 2144.94   682.2 2154.69   692.1 2168.98   731.8 2203.36
   761.6 2235.59   771.5 2251.04   781.4 2258.56   791.4 2261.66   831.1 2266.68
#Mann= 3 , 0 , 0
       0      .1       0   411.7    .045       0   436.7      .1       0
Bank Sta=411.7,436.7
XS Rating Curve= 0 ,0
Exp/Cntr=0.3,0.1

Type RM Length L Ch R = 1 ,51471.2 ,497.8,455.3,412.8
XS GIS Cut Line= 3
     1925120.788      282385.985     1925649.394      282440.127
     1925941.352      282182.051
#Sta/Elev= 30
       0  2102.8    39.4    2112      59  2107.1    68.9 2103.19    78.7 2095.02
   147.6    2066   157.4 2058.27   167.3 2053.61   216.5 2035.66   226.3 2029.41
     246 2005.32   275.5 1983.45     305 1975.77   334.6 1963.33   364.1 1959.49
   383.2 1959.49   393.6 1960.32   408.2 1966.69   442.8 1985.01   551.4 2004.28
   611.3  2022.6   651.3 2045.57   661.3 2047.97   691.2 2070.94   731.2 2095.24
   791.2 2126.08   801.1 2129.31   821.1 2129.85   861.1 2136.97     921 2153.42
#Mann= 3 , 0 , 0
       0      .1       0   383.2    .045       0   408.2      .1       0
Bank Sta=383.2,408.2
XS Rating Curve= 0 ,0
Exp/Cntr=0.3,0.1

Type RM Length L Ch R = 1 ,51015.1 ,344.9,336.7,330.1
XS GIS Cut Line= 3
     1925777.185      283067.276     1925859.723      282471.159
     1926011.975      282252.935
#Sta/Elev= 30
       0 2267.51    59.2 2233.72    78.9  2226.9    88.8 2218.91    98.7 2207.27
   118.4 2174.08   128.2 2161.27     148 2140.65   157.8 2133.24   167.7 2131.58
   187.4 2114.49     217 2093.25   246.6 2062.32   256.5 2061.14   266.4 2048.89
   305.8 1982.48   315.7 1973.05   335.4 1966.33   386.6 1954.96   411.6 1952.76
   414.4 1952.71   453.8 1962.53   473.6  1973.4   522.9 1994.34   542.6 1998.53
   621.5 2034.32   641.2 2039.86   729.9 2094.28   838.3 2119.77   867.9 2124.52
#Mann= 3 , 0 , 0
       0      .1       0   386.6    .045       0   411.6      .1       0
Bank Sta=386.6,411.6
XS Rating Curve= 0 ,0
Exp/Cntr=0.3,0.1

Type RM Length L Ch R = 1 ,50678.1 ,406.4,399.6,392.5
XS GIS Cut Line= 3
      1926232.59      283081.365     1926167.563      282678.001
     1926124.923      282265.438
#Sta/Elev= 30
       0 2250.57    19.9  2250.8    29.9 2247.32    39.9 2235.66    59.8 2204.41
    69.8 2193.91    79.7 2193.89    99.6 2184.06   129.6 2167.03   159.4 2145.24
   169.4 2143.72   179.4 2136.22   229.2  2088.1   259.1 2054.52     279 2042.38
   338.8 1971.91   348.8 1963.65   378.7 1951.47   396.1 1947.78   421.1 1947.57
   428.3 1947.54     458 1949.08   467.8 1953.32     537 1990.87   546.8 1991.85
   635.7 2044.97   645.6  2045.2   724.6 2088.13   734.5 2089.17   823.3 2120.45
#Mann= 3 , 0 , 0
       0      .1       0   396.1    .045       0   421.1      .1       0
Bank Sta=396.1,421.1
XS Rating Curve= 0 ,0
Exp/Cntr=0.3,0.1

Type RM Length L Ch R = 1 ,50278.1 ,394.4,399.7,403.8
XS GIS Cut Line= 3
     1926707.021      282926.593     1926544.913      282548.937
     1926400.637       282165.99
#Sta/Elev= 30
       0 2155.98    19.6 2152.54    29.4 2148.45    97.8 2115.35   117.4 2109.44
     137 2097.35   146.8  2094.1   195.7 2059.93   215.3 2052.47   264.2 2021.54
   303.3 1988.48   313.1 1982.55   322.9 1979.58   342.5 1965.27   371.8 1947.76
   381.6 1943.89   398.5  1942.4   401.2 1942.39   423.5 1942.56   460.9 1943.11
   500.8 1961.15   520.8 1966.24   530.8 1971.25   550.7 1984.74   600.6 2027.58
   610.6 2028.28   700.4 2077.23   720.4 2083.67   800.2 2150.62   820.2 2159.36
#Mann= 3 , 0 , 0
       0      .1       0   398.5    .045       0   423.5      .1       0
Bank Sta=398.5,423.5
XS Rating Curve= 0 ,0
Exp/Cntr=0.3,0.1

Type RM Length L Ch R = 1 ,49878.1 ,385.1,399.5,407.9
XS GIS Cut Line= 3
     1927006.997      282813.128     1926920.336      282412.897
     1926832.378      282012.959
#Sta/Elev= 30
       0 2103.07    69.9 2069.76    89.9 2065.31   159.8 2034.86   179.8 2031.19
   209.8 2020.47   249.7  1998.3   259.7 1993.56   269.7 1991.96   329.6 1954.58
   359.6 1944.55   369.6 1944.44     397 1938.18   409.5    1938     422 1938.02
   459.4 1938.45   469.4 1940.24   539.4 1969.09   559.3 1974.74   569.3 1982.73
   599.3  2015.1   629.2 2051.76   639.2 2060.89   649.2 2067.01   659.2 2079.37
   739.1 2196.07   749.1 2196.72     789 2250.77     799 2261.38     819 2268.72
#Mann= 3 , 0 , 0
       0      .1       0     397    .045       0     422      .1       0
Bank Sta=397,422
XS Rating Curve= 0 ,0
Exp/Cntr=0.3,0.1

Type RM Length L Ch R = 1 ,49478.1 ,378.7,379.7,386.9
XS GIS Cut Line= 3
     1927185.211      282840.146     1927310.065      282453.062
     1927350.184      282029.719
#Sta/Elev= 30
       0 2101.53     9.9 2100.66    89.3 2061.76   109.1 2055.95   198.4 2006.73
   208.3 2006.05   267.8 1971.82   287.7 1954.52     367 1933.34   394.2  1931.7
   419.2 1931.86   446.3 1932.14   456.2 1934.53     476 1944.17   495.7 1948.94
   535.3 1970.38   555.1  1978.1   574.8 1997.17   594.6 2009.01   614.4 2029.42
   634.2 2059.71   663.8 2113.14   683.6 2133.73   703.4 2172.88   723.2  2207.7
   752.8 2250.11   762.7 2255.95   782.5 2257.13   812.2 2257.05     832 2253.81
#Mann= 3 , 0 , 0
       0      .1       0   394.2    .045       0   419.2      .1       0
Bank Sta=394.2,419.2
XS Rating Curve= 0 ,0
Exp/Cntr=0.3,0.1

Type RM Length L Ch R = 1 ,49098.2 ,311.8,283.5,255.3
XS GIS Cut Line= 3
     1927513.671       282984.37     1927711.312      282440.127
      1927441.17      282053.207
#Sta/Elev= 30
       0  2168.3    49.9 2140.83    69.9 2133.98    79.9 2125.79   109.8  2090.7
   149.8 2048.88   159.7 2046.39   239.6  1982.5   249.6 1976.65   259.6 1974.95
   289.5 1951.42   309.5 1940.27   339.4 1929.44   358.8  1928.9   383.8  1929.3
   409.3 1934.89   439.3 1948.04   449.2  1948.3   459.2 1954.58   469.2 1966.82
   509.1 2024.81   539.1 2060.59   549.1 2067.02     569 2076.84     579 2079.01
   598.7 2090.21   687.2 2116.18   795.3 2133.63   942.8 2189.94  1050.9 2221.05
#Mann= 3 , 0 , 0
       0      .1       0   358.8    .045       0   383.8      .1       0
Bank Sta=358.8,383.8
XS Rating Curve= 0 ,0
Exp/Cntr=0.3,0.1

Type RM Length L Ch R = 1 ,48814.2 ,300.9,278.5,256.1
XS GIS Cut Line= 2
     1928181.106      282935.349     1927738.897      282381.941
#Sta/Elev= 30
       0 2192.17      20 2187.52    49.9 2173.41    89.8 2145.66   109.8 2125.45
   119.7 2120.66   179.6 2033.56   219.5 1963.06   229.5  1953.7   239.4 1940.88
   249.4 1931.34   259.4 1929.96   289.3  1937.8   329.2 1941.11   379.1 1949.09
   399.1 1941.93     419  1937.1   433.1 1928.93     439 1926.22   458.1 1925.37
   488.9 1926.71   498.9 1933.16   518.8 1955.87   548.8  1996.6   558.7  2007.6
   568.7 2015.47   618.6 2039.42   638.5 2051.08   658.5 2057.54   708.4 2068.54
#Mann= 3 , 0 , 0
       0      .1       0   433.1    .045       0   458.1      .1       0
#XS Ineff= 2 , 0
          378.63 1948.97
Permanent Ineff=
       F       F
Bank Sta=433.1,458.1
XS Rating Curve= 0 ,0
Exp/Cntr=0.3,0.1

Type RM Length L Ch R = 1 ,48535.5 ,585,583.4,581.7
XS GIS Cut Line= 2
     1928385.401      282374.183     1927694.934      282317.291
#Sta/Elev= 30
       0 2065.74    29.7 2076.56    49.5 2087.37    69.3  2094.5    79.2  2095.7
    89.1 2093.31   108.9 2081.94   128.7 2062.33     188 2022.91   207.8 2004.39
   267.2 1974.08   277.1 1968.23     287 1960.01   326.6 1940.14   346.4 1928.59
   363.8  1921.6   388.8 1920.79   425.6  1920.3   435.5 1921.72   445.4 1929.45
   465.2 1940.33     485 1959.18   494.9 1966.54   514.7 1977.66   524.6 1988.56
   593.8 2029.75   603.7 2039.76   613.6 2046.34     673  2075.7   692.8 2090.96
#Mann= 3 , 0 , 0
       0      .1       0   363.8    .045       0   388.8      .1       0
Bank Sta=363.8,388.8
XS Rating Curve= 0 ,0
Exp/Cntr=0.3,0.1

Type RM Length L Ch R = 1 ,47951.3 ,834.5,872.9,911.3
XS GIS Cut Line= 2
     1928160.418      281771.641     1927493.225      281756.125
#Sta/Elev= 30
       0 2065.73    49.8 2024.45    59.8 2015.25    69.7 1999.72   129.5 1950.82
   139.4 1942.16   149.4 1927.17   159.4 1921.86   169.3 1918.24   179.3 1916.01
   198.1 1915.06   199.2 1915.04   223.1 1915.08   239.1 1915.39     249 1917.28
     259 1921.14   298.8 1940.37   308.8 1950.72   378.5 1992.93   388.5 2005.18
   458.2 2048.13   468.2 2059.81   478.1 2066.61   537.9 2103.41   547.8 2114.64
   557.8  2121.5   617.6 2158.85   627.5 2169.98   637.5  2176.6   667.4 2192.27
#Mann= 3 , 0 , 0
       0      .1       0   198.1    .045       0   223.1      .1       0
Bank Sta=198.1,223.1
XS Rating Curve= 0 ,0
Exp/Cntr=0.3,0.1

Type RM Length L Ch R = 1 ,47077.7 ,380.6,392.5,404.4
XS GIS Cut Line= 2
     1928290.581      281481.576     1928150.074      280595.002
#Sta/Elev= 30
       0 2074.61    29.9 2065.62   109.7 2034.11   159.6  2019.9   219.4 1994.27
   249.3  1972.7   299.2 1927.18   329.1 1914.88     369 1911.28   458.8 1910.83
   498.5 1902.38   523.5 1901.26   548.6 1901.23   568.5 1901.99   588.4  1911.1
   598.4 1911.34   618.4 1924.76   668.2 1982.27   678.2 1991.74   688.2 1994.74
   698.2 2002.41   708.1 2013.52     748 2083.17     768 2109.21   787.9 2122.23
   807.9 2143.89   827.8 2161.25   857.7 2182.59   877.7 2189.94   897.6 2205.76
#Mann= 3 , 0 , 0
       0      .1       0   498.5    .045       0   523.5      .1       0
Bank Sta=498.5,523.5
XS Rating Curve= 0 ,0
Exp/Cntr=0.3,0.1

Type RM Length L Ch R = 1 ,46685   ,394.1,418.7,443.3
XS GIS Cut Line= 2
      1928393.19      281666.941      1928698.31      280582.072
#Sta/Elev= 30
       0 2141.58    79.8 2110.27   109.7  2095.2   119.7 2094.44   129.6 2090.04
   169.5 2071.74   209.4 2048.21   289.2 2022.57     369 2006.69     379 1997.12
   398.9 1969.08   408.9 1963.54   418.9  1954.1   438.8 1929.98   448.8  1920.3
   458.8 1915.56   528.6 1915.59   588.4 1906.54   678.2  1906.3   741.5 1898.07
   766.5 1897.61   797.8 1905.01   877.6 1985.65   887.6 1988.74   917.5 2015.33
   967.4 2073.76   987.3 2085.99  1077.1 2155.67  1087.1 2155.91    1127 2190.26
#Mann= 3 , 0 , 0
       0      .1       0   741.5    .045       0   766.5      .1       0
Bank Sta=741.5,766.5
XS Rating Curve= 0 ,0
Exp/Cntr=0.3,0.1

Type RM Length L Ch R = 1 ,46265.7 ,252,255.6,259.1
XS GIS Cut Line= 2
     1928553.492      281365.636     1929148.277       281109.62
#Sta/Elev= 30
       0  1972.1      10 1963.07    19.9 1952.58    29.9 1933.84    39.8 1922.25
    49.8 1914.73    59.8 1911.76   199.2 1910.98     259 1903.48   278.9  1898.6
   288.9 1893.62   298.9 1890.84   308.8 1890.44   323.4 1890.47   348.4 1891.21
   358.6 1894.36   368.6 1900.34   378.6 1911.45   418.4 1932.21   428.4  1938.6
   458.3 1965.36   468.2 1976.87   478.2 2000.45   547.9 2091.08   557.9  2106.7
   567.8 2125.39   597.7 2157.62   617.7  2176.2   637.6 2192.63   647.5 2203.64
#Mann= 3 , 0 , 0
       0      .1       0   323.4    .045       0   348.4      .1       0
Bank Sta=323.4,348.4
XS Rating Curve= 0 ,0
Exp/Cntr=0.3,0.1

Type RM Length L Ch R = 1 ,46010.1 ,538.9,547.5,556.1
XS GIS Cut Line= 2
     1928594.869      281575.103     1929146.022      281417.421
#Sta/Elev= 30
       0 1997.74    19.8 1979.29    69.2 1930.57    79.1 1914.62      89 1909.19
   108.7 1907.84   197.7 1908.73   237.2 1907.42   266.9 1904.04   296.5 1899.52
   306.4  1897.4   316.3 1893.98   326.2 1888.59     336  1885.8   340.9 1885.74
   345.9 1885.68   365.9 1886.45   375.6 1890.06   395.4 1903.26   405.2 1906.65
   454.7 1906.77   464.5  1909.6   474.4 1917.86   484.3 1929.57   494.2 1951.26
   504.1 1967.61   523.8 1993.39   533.7 2005.55   563.4 2039.49   573.3 2053.41
#Mann= 3 , 0 , 0
       0      .1       0   340.9    .045       0   365.9      .1       0
Bank Sta=340.9,365.9
XS Rating Curve= 0 ,0
Exp/Cntr=0.3,0.1

Type RM Length L Ch R = 1 ,45462.3 ,392.4,398.5,404.6
XS GIS Cut Line= 3
     1928491.428       281999.21     1928579.353      281994.038
     1929293.259      282017.169
#Sta/Elev= 30
       0 2118.96     9.8 2114.78    19.6 2106.68    29.4 2101.86    88.1  2076.6
   107.9 2056.06   167.4 2008.63   187.3 1985.03   246.8 1937.97   266.6 1914.69
   286.5 1899.78   296.4 1895.21   395.6 1893.29   455.1 1895.39     475 1892.38
   494.8  1885.4   514.7  1883.1   538.2 1883.15   563.2 1885.69     604 1902.68
   613.9 1910.88   623.8  1925.1   653.6 1974.26   663.5 1992.81   673.4 2021.41
   693.2 2046.24   703.2 2054.01   742.8 2076.08   752.8 2086.97   802.4 2114.58
#Mann= 3 , 0 , 0
       0      .1       0   538.2    .045       0   563.2      .1       0
#XS Ineff= 2 , 0
          456.49 1902.91
Permanent Ineff=
       F       F
Bank Sta=538.2,563.2
XS Rating Curve= 0 ,0
Exp/Cntr=0.3,0.1

Type RM Length L Ch R = 1 ,45063.5 ,383,394.3,405.7
XS GIS Cut Line= 2
     1928506.944      282281.086     1929245.552      282472.752
#Sta/Elev= 30
       0 2049.33    19.8 2027.94    89.2  1978.9    99.1 1965.27   168.5 1912.41
   178.4  1899.7   188.3 1892.58   198.2 1890.78   386.5 1888.95   406.3 1884.94
   426.1 1878.91     446  1877.7     450  1877.7     475  1877.7   495.5  1879.5
   505.4 1886.38   515.3 1896.55   525.2 1900.18     545  1903.3     555 1909.98
   584.7  1946.5   594.6 1970.16     664 2057.16   673.9 2077.11   683.8 2093.26
   703.6 2116.29   713.5 2124.76   723.4 2128.46   733.3 2127.35   763.1 2115.25
#Mann= 3 , 0 , 0
       0      .1       0     450    .045       0     475      .1       0
Bank Sta=450,475
XS Rating Curve= 0 ,0
Exp/Cntr=0.3,0.1

Type RM Length L Ch R = 1 ,44668.9 ,398.8,388.3,377.7
XS GIS Cut Line= 2
     1928481.084      282508.656     1929067.135      282970.411
#Sta/Elev= 30
       0 2000.49    39.8 1983.31    49.7 1973.84    69.6 1960.96    99.5 1938.23
   119.4    1926   139.3 1911.18   149.2 1898.88   159.2 1889.72   169.1 1886.42
   208.9 1887.11   308.4 1882.48   358.1 1875.05   382.6 1875.13   407.6 1875.37
   427.8 1875.54   437.7 1876.75   457.6 1883.06   477.5 1893.39   497.4 1899.65
   507.4 1900.36   547.1  1899.2   557.1  1900.2     567 1905.07     577 1913.31
   586.9 1919.34   656.6 1958.69   666.5  1965.2   676.5 1975.28   746.1 2007.94
#Mann= 3 , 0 , 0
       0      .1       0   382.6    .045       0   407.6      .1       0
Bank Sta=382.6,407.6
XS Rating Curve= 0 ,0
Exp/Cntr=0.3,0.1

Type RM Length L Ch R = 1 ,44280.3 ,250,246.9,243.9
XS GIS Cut Line= 2
     1928369.885      283015.516     1928973.701      283191.194
#Sta/Elev= 30
       0 2057.63    39.9 2026.98    59.9 2008.56    79.8 1975.03   119.8 1929.15
   149.7 1889.83   159.7 1882.99   199.6 1868.59   209.6 1867.22   218.5 1867.16
   219.6 1867.15   243.5 1867.55   259.5 1869.81   279.5 1876.32   289.5 1878.16
   319.4 1877.83   329.4 1879.46   349.4 1888.49   359.3 1891.64   369.3 1892.87
   419.2 1892.87   429.2 1891.65   489.1 1895.57   509.1 1898.22     519 1901.16
     529 1906.62     549  1920.2   578.9 1937.39   588.9 1944.52   628.8 1961.59
#Mann= 3 , 0 , 0
       0      .1       0   218.5    .045       0   243.5      .1       0
Bank Sta=218.5,243.5
XS Rating Curve= 0 ,0
Exp/Cntr=0.3,0.1

Type RM Length L Ch R = 1 ,44033.3 ,564.1,554.8,545.4
XS GIS Cut Line= 3
     1928118.637      283246.485     1928522.026      283316.969
     1928925.414      283387.453
#Sta/Elev= 30
       0 2100.01      10 2093.06    79.9  2054.5    99.9 2039.22   119.8    2027
   149.8 2004.45   159.8 1995.82   179.8 1975.77   239.7 1938.37   249.7 1930.75
   259.7  1920.4   319.6  1884.9   329.6 1880.58   349.6 1875.96   369.6    1867
   379.5 1864.12   389.5 1863.68   397.4 1863.78   422.4 1864.08   439.5 1865.68
   459.4 1876.44   469.4 1880.25   499.4 1880.51   549.3 1891.91   719.1 1896.59
   729.1 1898.14   739.1 1903.91   749.1 1911.84   759.1  1917.1     819 1945.29
#Mann= 3 , 0 , 0
       0      .1       0   397.4    .045       0   422.4      .1       0
Bank Sta=397.4,422.4
XS Rating Curve= 0 ,0
Exp/Cntr=0.3,0.1

Type RM Length L Ch R = 1 ,43478.1 ,405.4,399.5,393.7
XS GIS Cut Line= 3
      1928095.79      283930.036     1928499.855      283863.585
     1928903.559      283794.853
#Sta/Elev= 30
       0 2024.96      20 2013.43      40  1996.4    69.9 1981.25   119.8 1963.41
   159.8 1954.95   179.8  1947.2   189.8  1941.7   209.7 1923.06   239.7 1903.03
   289.6 1878.64   349.6 1865.83   369.5 1858.81   379.5 1858.22     397 1858.25
     422 1858.39   439.5 1858.65   519.4 1880.29   549.3 1900.02   559.3 1910.43
   569.3 1927.42   579.3 1950.25   609.3 2025.93   619.2 2046.24   649.2 2062.75
   729.1 2083.91   759.1 2100.15   769.1 2106.93     779 2116.59     819  2130.3
#Mann= 3 , 0 , 0
       0      .1       0     397    .045       0     422      .1       0
Bank Sta=397,422
XS Rating Curve= 0 ,0
Exp/Cntr=0.3,0.1

Type RM Length L Ch R = 1 ,43078.1 ,400.6,399.8,398.5
XS GIS Cut Line= 3
      1928247.72      284391.634     1928628.125      284240.165
     1929008.831      284088.679
#Sta/Elev= 30
       0 2075.97      40 2041.99    49.9 2031.42    59.9 2017.11    69.9 2008.99
    89.9 1995.03   129.8 1972.18   149.8 1956.87   189.8 1938.94   219.7 1922.92
   229.7 1913.39   239.7 1907.52   319.6 1867.76   339.6 1864.85   369.5 1855.21
     397 1853.93   419.4  1853.7     422 1853.89   429.4 1854.42   439.4    1858
   479.4 1885.62   489.4 1894.92   559.4 1925.61   579.3 1937.48   649.3 1965.93
   659.3 1971.66   709.3  1993.2   739.2 2008.17   749.2 2016.22   819.2 2049.42
#Mann= 3 , 0 , 0
       0      .1       0     397    .045       0     422      .1       0
Bank Sta=397,422
XS Rating Curve= 0 ,0
Exp/Cntr=0.3,0.1

Type RM Length L Ch R = 1 ,42678.1 ,388,399.5,412.3
XS GIS Cut Line= 3
     1928418.152      284765.656     1928794.244      284603.709
     1929167.095      284433.966
#Sta/Elev= 30
       0 2136.78    49.9 2099.85    59.9 2087.49    89.9 2063.76   159.8 2020.35
   189.8 1997.64   219.7 1970.77   239.7 1944.63   259.7 1923.63   289.6    1895
   309.6 1878.19   319.6  1867.8   329.6 1862.82   359.5 1852.09   389.5 1849.55
     397  1849.6     422 1850.24   479.4 1860.26   529.4 1875.68   569.4 1896.54
   579.3 1903.11   609.3 1912.69   639.3  1927.3   659.3 1938.06   669.3 1946.07
   699.2 1963.58   749.2 1988.78   769.2 2000.44   799.2 2013.82   819.2 2016.41
#Mann= 3 , 0 , 0
       0      .1       0     397    .045       0     422      .1       0
Bank Sta=397,422
XS Rating Curve= 0 ,0
Exp/Cntr=0.3,0.1

Type RM Length L Ch R = 1 ,42278.1 ,391.5,399.8,407.3
XS GIS Cut Line= 3
     1928476.055      284984.136     1928885.711      284988.833
     1929294.874      285004.626
#Sta/Elev= 30
       0 2097.85      60 2062.76   109.9 2023.02   139.9 2004.63   159.9 1984.86
   179.9 1968.06   199.8 1948.99   219.8 1934.05   239.8 1915.91   279.8 1895.68
   299.8 1883.54   319.8 1864.89   329.7 1859.82   369.7 1846.76   389.7 1844.68
   397.2  1844.7   422.2 1846.08   429.7  1848.2   469.6 1869.01   489.6 1882.25
   549.5 1909.61   569.5 1923.24   629.4 1951.34   639.4 1957.45   649.4 1965.92
   709.3 1992.95   729.3 2005.13   789.2 2028.03   809.2 2038.94   819.2  2042.4
#Mann= 3 , 0 , 0
       0      .1       0   397.2    .045       0   422.2      .1       0
Bank Sta=397.2,422.2
XS Rating Curve= 0 ,0
Exp/Cntr=0.3,0.1

Type RM Length L Ch R = 1 ,41878.1 ,396.9,399.9,402.8
XS GIS Cut Line= 3
     1928418.987      285253.594     1928808.599      285379.661
     1929198.211      285505.727
#Sta/Elev= 30
       0 2008.37      40 1989.42    69.9 1968.19   139.8 1929.78   149.8 1919.96
   179.8 1902.75   239.7 1874.11   299.6 1854.81   319.6 1846.68   339.6 1845.46
   359.6 1839.78   379.5 1838.55     397 1838.68     422 1838.86   439.5 1839.21
   449.4  1841.1   459.4 1845.19   479.4 1857.78   489.4 1867.64   549.3 1904.27
   559.3 1911.29   569.3 1923.99   579.3 1932.98   619.2 1965.12   639.2 1977.14
   659.2 1993.97   729.1 2041.65   739.1 2054.96     809 2107.12     819 2115.67
#Mann= 3 , 0 , 0
       0      .1       0     397    .045       0     422      .1       0
Bank Sta=397,422
XS Rating Curve= 0 ,0
Exp/Cntr=0.3,0.1

Type RM Length L Ch R = 1 ,41478.1 ,404.9,399.8,393.7
XS GIS Cut Line= 3
     1928287.608      285584.162     1928661.467      285751.255
     1929035.325      285918.348
#Sta/Elev= 30
       0 1965.57      20 1957.95      40 1947.03    99.9  1928.6   129.8 1912.78
   199.8 1903.34   219.7  1896.9   259.7 1873.74   319.6 1846.48   349.6 1842.69
   389.5 1831.19     397 1831.24     422 1831.35   439.5 1833.82   449.4 1839.04
   459.4 1845.55   479.4 1864.91   519.4 1893.02   549.3 1925.16   559.3 1942.02
   569.3  1955.1   589.3 1972.89   649.2 2039.02   659.2 2055.76   669.2 2068.24
   739.1 2129.81   749.1 2141.21   769.1  2152.3     789 2167.42     819 2177.32
#Mann= 3 , 0 , 0
       0      .1       0     397    .045       0     422      .1       0
Bank Sta=397,422
XS Rating Curve= 0 ,0
Exp/Cntr=0.3,0.1

Type RM Length L Ch R = 1 ,41078.1 ,421,399.6,381.5
XS GIS Cut Line= 3
     1928136.546      286032.522     1928534.318      286129.484
       1928936.4      286209.448
#Sta/Elev= 30
       0 2011.65      10 2008.13      30 1996.42    89.9  1967.5    99.9 1961.78
   109.8 1952.96   179.7 1921.14   189.7 1912.89   199.7 1907.68   269.6 1875.64
   289.6 1861.26   339.5 1837.43   359.5 1830.49   369.5  1828.3   396.9 1828.33
   421.9 1828.46   479.4 1832.35   489.4 1834.52   499.4 1839.38   519.4 1853.01
   529.4 1866.64   599.4 1914.96   609.4 1927.54   619.4 1935.52   679.4 1972.59
   689.4 1982.37   699.4  1990.4   759.4 2024.27   779.4 2041.45   819.4  2065.9
#Mann= 3 , 0 , 0
       0      .1       0   396.9    .045       0   421.9      .1       0
Bank Sta=396.9,421.9
XS Rating Curve= 0 ,0
Exp/Cntr=0.3,0.1

Type RM Length L Ch R = 1 ,40678.1 ,390,399.5,409.6
XS GIS Cut Line= 3
     1928219.335      286727.427     1928568.011      286517.832
     1928948.351      286328.928
#Sta/Elev= 30
       0  2070.8    19.8    2067    39.7 2057.63   119.1 2038.65   138.9 2023.55
   158.8 2015.35   168.7 2008.81   208.4  1980.1   218.3 1969.71   248.1 1936.82
   287.8 1885.87   307.6 1865.01   317.5 1848.49   327.4 1838.04   347.3 1825.48
   357.2 1822.42   377.1 1820.79   394.3 1820.88   419.3 1821.64   515.5 1829.38
   535.2 1833.28   545.1 1837.77   574.7 1860.76   594.5  1879.7   663.6  1921.9
   683.4 1939.83   742.6 1980.11   752.5 1987.64   772.2  2009.1   831.5 2054.16
#Mann= 3 , 0 , 0
       0      .1       0   394.3    .045       0   419.3      .1       0
Bank Sta=394.3,419.3
XS Rating Curve= 0 ,0
Exp/Cntr=0.3,0.1

Type RM Length L Ch R = 1 ,40278.1 ,390.1,399.7,403.9
XS GIS Cut Line= 3
      1928350.87      286936.498     1928765.322      286854.333
     1929170.815       286817.06
#Sta/Elev= 30
       0 2041.91      59  2005.4    78.6 1987.83   108.1 1971.76   137.6 1952.26
   157.2 1934.63     226 1893.07   235.8 1881.04   304.6 1843.92   324.3 1828.64
   353.7 1819.85   373.4 1816.14     393 1814.96     410 1815.03     435  1815.1
   452.3 1816.33   472.2 1822.81   482.1 1830.78   511.9  1846.1   531.8 1859.43
   551.6 1876.68   561.6 1891.95   631.1 1952.53     641 1969.48   710.5  2027.7
   720.5 2043.86   730.4  2053.2     790 2097.54   799.9 2110.14   829.7 2131.58
#Mann= 3 , 0 , 0
       0      .1       0     410    .045       0     435      .1       0
Bank Sta=410,435
XS Rating Curve= 0 ,0
Exp/Cntr=0.3,0.1

Type RM Length L Ch R = 1 ,39878.1 ,416,399.5,386.2
XS GIS Cut Line= 3
     1928319.555      287186.389     1928723.553      287250.748
     1929134.662      287274.784
#Sta/Elev= 30
       0 2052.58      10 2047.03      20 2037.12    29.9 2030.08    89.8 1997.26
   109.8 1970.66   169.6 1929.15   189.6 1908.06   249.4  1869.3   269.4 1851.28
   319.3 1821.32   349.2 1807.51   396.6 1806.95   421.6 1806.77   438.5 1806.67
   458.1 1809.41   487.5 1827.49   497.3 1834.09   507.1 1847.07   575.8 1896.62
   585.6 1916.26   595.4 1940.35   605.2 1961.34     615 1974.42     664  2007.5
   683.6 2026.02   742.5 2067.94   762.1 2085.38   791.5 2099.18   820.9 2117.98
#Mann= 3 , 0 , 0
       0      .1       0   396.6    .045       0   421.6      .1       0
Bank Sta=396.6,421.6
XS Rating Curve= 0 ,0
Exp/Cntr=0.3,0.1
